--- KENSCK.prj (project) ---

Proj Title=KENSCK
Current Plan=p01
Default Exp/Contr=0,0
English Units
Geom File=g01
Flow File=f01
Plan File=p01
Background Map Layer=Inundation Boundary (01pct Value_0)
Background Map Layer=Inundation Boundary (01pct Value_0)
BEGIN DESCRIPTION:
----------MODEL BY WOOD PLC 2021----------
Stream Name: Kens Creek
Flood Zone: Approximate
Pocahontas County, WV
HEC-RAS Version: RAS 6.1
Vertical Datum: NAVD88
Projection: NAD 1983 StatePlane West Virginia S FIPS 4702 (US Feet)
Terrain: 1-meter LIDAR (FEMA Region III 3DEP collected 2016-2018)
Land Use: 2019 NLCD
Hydrologic Method:
WV SIR2010-5033 regression equations
END DESCRIPTION:
DSS Export Rating Curves= 0
DSS Export Rating Curve Sorted= 0
DSS Export Volume Flow Curves= 0
DXF OffsetX= 0
DXF OffsetY= 0
DXF ScaleX= 0
DXF ScaleY= 0

--- KENSCK.p01 (plan) ---

Plan Title=Floodplain
Program Version=6.00
Short Identifier=Floodplain
Geom File=g01
Flow File=f01
Subcritical Flow
K Sum by GR= 0
Std Step Tol= 0.01
Critical Tol= 0.01
Num of Std Step Trials= 20
Max Error Tol= 0.3
Flow Tol Ratio= 0.001
Split Flow NTrial= 30
Split Flow Tol= 0.02
Split Flow Ratio= 0.02
Log Output Level= 0
Friction Slope Method= 1
Unsteady Friction Slope Method= 2
Unsteady Bridges Friction Slope Method= 1
Parabolic Critical Depth
Global Vel Dist= 0 , 0 , 0
Global Log Level= 0
CheckData=False
Encroach Param=-1 ,0,0, 0
Mapping Interval=1HOUR
Computation Time Step Use Courant=        0
Computation Time Step Use Time Series=    0
Computation Time Step Count To Double=0
Computation Time Step Max Doubling=0
Computation Time Step Max Halving=0
Computation Time Step Residence Courant=0
Run HTab= 0
Run UNet= 0
Run Sediment= 0
Run PostProcess= 0
Run WQNet= 0
Run RASMapper=-1
UNET Theta= 0
UNET Theta Warmup= 0
UNET ZTol= 0
UNET ZSATol= 0
UNET MxIter= 0
UNET Max Iter WO Improvement= 0
UNET MaxInSteps= 0
UNET DtIC= 0
UNET DtMin= 0
UNET MaxCRTS= 0
UNET WFStab= 0
UNET SFStab= 0
UNET WFX= 1
UNET SFX= 1
UNET Gravity=32.174
UNET 1D Methodology=Finite Difference
UNET DSS MLevel= 1
UNET Pardiso=0
UNET DZMax Abort= 0
UNET Use Existing IB Tables= 0
UNET Froude Reduction=False
UNET Froude Limit= 0
UNET Froude Power= 0
UNET D1 Cores= 0
UNET WindReference=Eulerian
UNET WindDragFormulation=Hsu (1988)
UNET D2 Coriolis=0
UNET D2 Cores= 0
UNET D2 Theta= 1
UNET D2 Theta Warmup= 1
UNET D2 Z Tol= 0.01
UNET D2 Volume Tol= 0.01
UNET D2 Max Iterations= 20
UNET D2 Equation= 0
UNET D2 RampUpFraction=0.1
UNET D2 TimeSlices= 1
UNET D2 Turbulence Formulation=Non-Conservative (original)
UNET D2 Eddy Viscosity=0.3
UNET D2 Transverse Eddy Viscosity=0.1
UNET D2 Smagorinsky Mixing=0
UNET D2 BCVolumeCheck=0
UNET D2 Cores=0
UNET D2 SolverType=PARDISO (Direct)
UNET D2 Minimum Iterations= 2147483647
UNET D2 Maximum Iterations= 2147483647
UNET D2 Restart Number= 10
UNET D2 Relaxation Coeff=1.3
UNET D2 SOR Precondition Iterations= 10
UNET D2 ILUT Maximum Fill= 8
UNET D2 ILUT Tolerance=1E-08
UNET D1D2 MaxIter= 0
UNET D1D2 ZTol=0.01
UNET D1D2 QTol=0.1
UNET D1D2 MinQTol=1
Write IC File= 0
Write IC File at Fixed DateTime=0
Write IC File at Sim End=0
Echo Input=False
Echo Parameters=False
Echo Output=False
Write Detailed= 0
HDF Write Warmup=0
HDF Write Time Slices=0
HDF Flush=0
HDF Compression= 1
HDF Chunk Size= 1
HDF Spatial Parts= 1
HDF Use Max Rows=0
HDF Fixed Rows= 1
Calibration Method= 0
Calibration Iterations= 20
Calibration Max Change=0.05
Calibration Tolerance=0.2
Calibration Maximum=1.5
Calibration Minimum=0.5
Calibration Optimization Method= 1
WQ AD Non Conservative
WQ ULTIMATE=-1
WQ Max Comp Step=1HOUR
WQ Output Interval=15MIN
WQ Output Selected Increments= 0
WQ Output face flow=0
WQ Output face velocity=0
WQ Output face area=0
WQ Output face dispersion=0
WQ Output cell volume=0
WQ Output cell surface area=0
WQ Output cell continuity=0
WQ Output cumulative cell continuity=0
WQ Output face conc=0
WQ Output face dconc_dx=0
WQ Output face courant=0
WQ Output face peclet=0
WQ Output face adv mass=0
WQ Output face disp mass=0
WQ Output cell mass=0
WQ Output cell source sink temp=0
WQ Output nsm pathways=0
WQ Output nsm derived pathways=0
WQ Create Restart=0
WQ Fixed Restart=0
WQ System Summary=0
WQ Write To DSS=0
Sorting and Armoring Iterations= 10
XS Update Threshold= 0.02
Bed Roughness Predictor= 0
Hydraulics Update Threshold= 0.02
Energy Slope Method= 1
Volume Change Method= 1
Sediment Retention Method= 0
Sediment TS Multiplier= 1
Warm Up Method= 0
XS Weighting Method= 0
Number of US Weighted Cross Sections= 1
Number of DS Weighted Cross Sections= 1
Upstream XS Weight=0
Main XS Weight=1
Downstream XS Weight=0
Number of DS XS's Weighted with US Boundary= 1
Upstream Boundary Weight= 1
Weight of XSs Associated with US Boundary= 0
Number of US XS's Weighted with DS Boundary= 1
Downstream Boundary Weight= 0.5
Weight of XSs Associated with DS Boundary= 0.5
Percentile Method= 0
Sediment Output Level= 3
Mass or Volume Output= 0
Output Increment Type= 1
Profile and TS Output Increment= 1
Transport Output Increment 1
XS Output Flag= 0
XS Output Increment= 10
Read HDF5 Sediment Hotstart= 0
Sediment Hotstart Type= 0
Write Gradation File= 0
Read Gradation Hotstart= 0
Write HDF5 File= 1
Write Binary Output= 1
Write DSS Sediment File= 0
DSS Sediment Output Type= 1
SV Curve= 0
Specific Gage Flag= 0
Subcell Erosion Methods= 0
Subcell Deposition Methods= 0
Advection Scheme= 1
Matrix Solver= 0
Implicit Weighting Factor= 1
Maximum Outer Loop Convergence Iterations= 5
Convergence Maximum Absolute= 0.001
Convergence RMSE= 0.0001
Grain Fractions Max Abs Error= 0.001
Max Subgrid Regions= 1
Max Subgrid Length Scale= 3.402823E+38
Initial Layer Thickness= 3.402823E+38
Min Layer Thickness= 3.402823E+38
Max Layer Thickness= 3.402823E+38
Number of Layers= 5

--- KENSCK.f01 (steady flow) ---

Flow Title=Flow
Program Version=6.00
Number of Profiles= 6
Profile Names=01pct,10pct,04pct,02pct,0_2pct,01plus
River Rch & RM=KENSCK,Main,6928
     577     305     406     489     807     854
River Rch & RM=KENSCK,Main,5008
     651     346     458     552     907     962
River Rch & RM=KENSCK,Main,3446
     737     393     521     625    1020    1090
Boundary for River Rch & Prof#=KENSCK,Main            , 1
Up Type= 0
Dn Type= 3
Dn Slope=0.06704
Boundary for River Rch & Prof#=KENSCK,Main            , 2
Up Type= 0
Dn Type= 3
Dn Slope=0.06704
Boundary for River Rch & Prof#=KENSCK,Main            , 3
Up Type= 0
Dn Type= 3
Dn Slope=0.06704
Boundary for River Rch & Prof#=KENSCK,Main            , 4
Up Type= 0
Dn Type= 3
Dn Slope=0.06704
Boundary for River Rch & Prof#=KENSCK,Main            , 5
Up Type= 0
Dn Type= 3
Dn Slope=0.06704
Boundary for River Rch & Prof#=KENSCK,Main            , 6
Up Type= 0
Dn Type= 3
Dn Slope=0.06704
DSS Import GetInterval= 0
DSS Import GetPeak= 0
DSS Import FillOption= 0

--- KENSCK.g01 (geometry) ---

Geom Title=Geometry
Program Version=6.10

River Reach=KENSCK          ,Main
Reach XY= 30
2182484.07099999      485936.5222182453.94000001486117.758000016
     2182546.443486218.3139999962182665.73999999486528.192000017
2182565.95900001486928.4190000152182590.42250006487374.076000005
2182631.38633893487496.7260810582182535.69400002487676.516000018
2182516.72400002487952.0150000162182441.78528516488008.989307791
2182394.57799999488186.6020000132182537.74000002488469.578000009
2182499.85900001488763.0370000152182733.15000002488994.927000016
2182701.79900004489079.3110000042182703.58300002 489337.13500002
2182803.53700002489572.1880000082182650.65500002489891.017000005
2182569.31438817 490168.595804142182757.99750008490342.264499992
2182698.55250002490495.488500014     2182685.355490719.307000011
      2182777.55491026.9920000142182674.47600003 491167.56400001
2182663.82224052491324.0735287522182740.79184683 491552.63841027
2182733.27749999491646.0330000072182663.65700002491841.999000013
2182499.11900003492016.4839999972182412.51139815492425.112980902

Type RM Length L Ch R = 1 ,6928    ,164.9,171.8,177.3
XS GIS Cut Line= 4
2182295.34152173486225.3423466242182447.54293706486212.713091871
2182587.12388626486085.6032021692182733.01506852486031.113724456
#Sta/Elev= 30
       0 3378.97    24.9  3367.9      45 3362.03      61 3358.83    81.1  3353.2
    93.2 3347.87   113.2 3336.94   129.3 3332.83   145.3 3330.87   181.2 3314.33
   189.7 3308.75   198.1 3301.16   209.5 3292.83   213.1 3290.95   220.8  3289.4
   226.5 3289.11   237.8 3289.46   256.4 3292.33     278 3307.55   282.7 3310.39
   288.8 3312.21   314.2 3316.23   346.9  3319.5     380 3325.05   393.9  3328.8
   410.9 3331.24   423.8 3334.91   432.8 3335.66   462.2 3345.05   497.2 3351.91
#Mann= 3 ,-1,0
       0      .1       0   220.8    .045       0   237.8      .1       0
Bank Sta=220.8,237.8
XS Rating Curve= 0 ,0
Exp/Cntr(USF)=0,0
Exp/Cntr=0.3,0.1

Type RM Length L Ch R = 1 ,6756    ,97.8,98.8,100
XS GIS Cut Line= 3
2182348.40574539486333.7949368442182508.18033123486342.838781326
2182809.64181394486211.703036348
#Sta/Elev= 30
       0 3363.06    27.8  3355.6    47.8 3347.89    55.9 3347.13    79.9 3340.71
   116.7 3328.01   147.1 3320.03   168.7 3310.73   181.8  3303.4   190.6 3299.28
   203.6 3288.54   221.1  3276.1   229.8 3275.72   240.3 3275.97   252.5 3278.21
   260.4 3281.81   269.1 3282.81   273.4  3284.2   286.5 3293.79   312.7 3305.81
   321.4 3307.72   347.6 3311.31     365 3315.24   377.1 3320.26   398.4 3327.32
     413 3333.23   426.1 3336.62   439.2 3342.92   447.9 3344.01   488.8 3358.04
#Mann= 3 ,-1,0
       0      .1       0   221.1    .045       0   240.3      .1       0
Bank Sta=221.1,240.3
XS Rating Curve= 0 ,0
Exp/Cntr(USF)=0,0
Exp/Cntr=0.3,0.1

Type RM Length L Ch R = 1 ,6658    ,192.6,201.9,213.6
XS GIS Cut Line= 3
2182360.69671422486442.5072267752182534.23672074486433.098431241
2182809.18263468486334.828788996
#Sta/Elev= 30
       0 3358.46      35 3350.72    76.8  3338.4   103.6 3332.98   119.7 3327.08
   135.7 3322.81   167.5  3312.7   180.1 3306.86   188.6 3301.65   201.3 3295.88
   215.9  3282.3   228.4 3274.16     233  3272.7   247.2 3271.39   260.8 3270.32
   269.3 3271.42   286.3 3275.13     299 3275.53   307.5 3280.12   341.5 3289.45
   347.4 3293.03   358.5 3301.51   362.8 3303.73   379.7 3316.08   392.5 3321.69
     401 3328.12     418 3335.07   434.9 3347.51   456.2 3356.07   465.8 3358.95
#Mann= 3 ,-1,0
       0      .1       0   247.2    .045       0   269.3      .1       0
Bank Sta=247.2,269.3
XS Rating Curve= 0 ,0
Exp/Cntr(USF)=0,0
Exp/Cntr=0.3,0.1

Type RM Length L Ch R = 1 ,6456    ,126.3,123.9,120.5
XS GIS Cut Line= 3
2182397.27041944486558.0357630982182585.05300932486565.920278529
2182851.27011038486674.786764753
#Sta/Elev= 30
       0 3348.97    22.9 3342.05    42.9  3337.6    59.6 3332.43      71  3331.8
      79 3330.06     111 3316.93     147 3299.14   183.1 3287.32   204.3 3279.33
   221.6 3271.26   232.7 3264.25   238.8 3259.41   243.2 3257.89   251.8 3257.05
   260.5 3255.12   270.5 3256.99   277.8 3257.92   297.1 3256.82   312.3 3259.16
   316.6 3262.88   325.3  3272.8   346.2    3286   349.3 3287.33   370.7 3292.67
   410.6 3300.97     442 3308.75   454.9 3312.73   463.6 3314.31   475.6 3318.08
#Mann= 3 ,-1,0
       0      .1       0   251.8    .045       0   270.5      .1       0
Bank Sta=251.8,270.5
XS Rating Curve= 0 ,0
Exp/Cntr=0.3,0.1

Type RM Length L Ch R = 1 ,6332    ,128.5,129,130.8
XS GIS Cut Line= 2
2182388.69406177486668.1782842592182826.47163173486752.121070733
#Sta/Elev= 30
       0 3348.97    27.8  3340.8    52.4 3332.28    68.7 3328.16    89.1 3324.59
   101.3 3323.77   121.7  3318.1   137.9 3310.83   162.4 3296.73   174.5 3290.71
   190.9 3276.21     199 3263.58   207.2 3259.17   223.5 3248.38   229.4 3247.53
     239 3247.29     252  3247.5   256.1 3248.99   264.2 3254.34   276.4 3256.16
   280.7 3259.12   288.6 3266.75   292.7 3268.52   321.2 3276.36   333.4 3278.85
   345.7  3279.9     366  3285.6   410.5 3291.46   424.2 3295.27   445.8 3303.46
#Mann= 3 ,-1,0
       0      .1       0   229.4    .045       0     252      .1       0
Bank Sta=229.4,252
XS Rating Curve= 0 ,0
Exp/Cntr(USF)=0,0
Exp/Cntr=0.3,0.1

Type RM Length L Ch R = 1 ,6203    ,184.4,180,176.3
XS GIS Cut Line= 2
2182385.50636101486782.9355113372182838.15986782486904.068139918
#Sta/Elev= 30
       0 3349.56    23.5 3339.29    31.7 3336.87    44.2 3330.51    85.7 3315.32
   111.8 3303.27     127 3291.77   139.4 3283.52   147.7  3275.5   160.1  3267.5
   172.5 3254.84   189.1 3242.03   193.63239.588   204.1  3238.5   216.3 3239.63
   226.7 3244.04   234.6 3246.01   247.1 3246.59   259.5 3245.59   271.9 3246.87
   287.2 3259.66   292.6 3262.52   300.9  3263.8   309.2 3263.54     334 3265.69
   371.3  3271.6   383.7 3275.85   416.8 3284.78     445 3295.35   468.6 3301.17
#Mann= 3 ,0,0
       0      .1       0   193.6    .045       0   216.3      .1       0
Bank Sta=193.6,216.3
XS Rating Curve= 0 ,0
Exp/Cntr(USF)=0,0
Exp/Cntr=0.3,0.1

Type RM Length L Ch R = 1 ,6023    ,155.6,153.5,152.4
XS GIS Cut Line= 2
2182340.67246067487012.2444175222182856.17159609487015.259032349
#Sta/Elev= 30
       0 3354.54    39.5 3342.26    63.5 3332.98    79.5 3323.96    91.5 3320.73
   107.2  3309.8   119.7 3298.92   127.5 3294.23   135.5 3286.85   147.4 3278.34
   175.6 3263.64   191.7 3251.91  214.42 3231.69   227.5 3230.47   235.1 3231.69
   243.5 3232.06   260.1 3237.26   275.5 3238.42   287.5 3243.36   311.5 3247.45
   327.5 3253.56   350.4 3259.31   375.5  3261.8   403.5 3267.45   431.5 3271.43
   447.5 3276.99   479.5 3294.39   495.5 3301.48   507.5 3309.17   515.5 3312.05
#Mann= 3 ,0,0
       0      .1       0  214.42    .045       0   235.1      .1       0
Bank Sta=214.42,235.1
XS Rating Curve= 0 ,0
Exp/Cntr(USF)=0,0
Exp/Cntr=0.3,0.1

Type RM Length L Ch R = 1 ,5869    ,115.9,116.4,117
XS GIS Cut Line= 3
 2182335.5657159487075.1414136172182525.76519411487171.835003098
 2182781.8438212487147.395963998
#Sta/Elev= 30
       0 3349.06     9.7 3346.09    23.1 3340.17    34.7  3337.1    63.5  3323.8
    94.9 3311.57   103.9  3305.6   126.3 3295.31   148.8 3282.12   159.6 3277.91
   184.7 3259.08   198.3 3252.03   210.2 3243.01   223.8 3234.79   247.9  3225.8
     256 3224.12     264 3223.59     272 3223.03   280.1 3223.64   304.2 3229.31
   308.2 3233.81   312.2 3237.06   324.1 3241.06   344.4 3246.36   356.4 3248.58
   396.6 3259.66     413 3262.09   436.8 3271.91   460.9 3279.02   470.6 3283.66
#Mann= 3 ,-1,0
       0      .1       0     264    .045       0   280.1      .1       0
Bank Sta=264,280.1
XS Rating Curve= 0 ,0
Exp/Cntr(USF)=0,0
Exp/Cntr=0.3,0.1

Type RM Length L Ch R = 1 ,5753    ,216.7,217,216.5
XS GIS Cut Line= 3
2182387.63149485487233.463884306 2182555.5170678487284.467096341
2182831.78446631487266.403458745
#Sta/Elev= 30
       0 3299.35     8.9 3294.32    17.3 3291.72      34 3284.81    64.3 3269.59
   100.9 3254.39   121.8 3247.99   134.9 3242.72   155.2 3233.21   186.7 3221.55
   204.2 3217.96   219.8 3217.55   228.2 3218.01   256.3    3221   264.3 3224.57
   280.3 3225.25   288.4 3227.19   296.4 3231.65   312.4 3243.55   320.4  3248.1
   328.4  3250.8   339.9 3257.77   359.8 3266.37   380.6 3278.14   392.6 3282.23
   404.6 3287.75   416.6 3295.53   420.6 3297.34   428.7 3298.23   452.3 3310.53
#Mann= 3 ,-1,0
       0      .1       0   204.2    .045       0   228.2      .1       0
Bank Sta=204.2,228.2
XS Rating Curve= 0 ,0
Exp/Cntr(USF)=0,0
Exp/Cntr=0.3,0.1

Type RM Length L Ch R = 1 ,5536    ,119.6,129.3,138.4
XS GIS Cut Line= 3
2182344.50433784487387.9834682892182512.27473628487497.099032823
2182838.26620689487479.691188543
#Sta/Elev= 30
       0 3292.97    53.5 3272.06    90.3 3258.94   128.4 3248.05     138 3243.95
   157.1 3234.07   176.2 3227.08     200 3221.51   220.1 3218.93   236.1 3215.19
   248.1 3214.14   256.1 3211.91   296.2 3208.77   304.2 3206.26   310.1 3205.57
   316.2    3205   329.3 3205.59   336.2 3206.48   340.7 3210.39   356.3 3226.96
   364.3 3233.06   376.3 3240.28   384.3 3247.05   424.4 3267.17   454.7 3286.72
   485.2 3300.95   500.4 3309.37   508.5 3312.02   516.5 3316.41   526.6 3320.59
#Mann= 3 ,0,0
       0      .1       0   310.1    .045       0   329.3      .1       0
Bank Sta=310.1,329.3
XS Rating Curve= 0 ,0
Exp/Cntr=0.3,0.1

Type RM Length L Ch R = 1 ,5407    ,145,138.2,133
XS GIS Cut Line= 3
2182318.17297834487467.9083930682182476.14781694487536.441595107
2182707.30217636487695.578013401
#Sta/Elev= 30
       0 3293.52    13.2    3286      24 3283.69    57.2 3272.63    93.7 3256.09
   111.2 3249.24   124.3 3245.68   136.3 3240.57   150.4 3232.97   177.1  3220.6
   194.7 3217.88   201.5 3215.54   215.9 3212.58   235.4  3209.5   245.1 3206.32
   264.8 3204.93   273.4 3200.96     282 3200.49   290.7 3199.61   296.4 3200.39
   310.8 3201.26   327.6  3204.7   332.5 3207.78   345.3 3218.04   351.1 3221.47
     377  3233.2   402.8 3246.99   413.3 3251.08   424.8 3254.01   452.8 3263.97
#Mann= 3 ,0,0
       0      .1       0     282    .045       0   296.4      .1       0
Bank Sta=282,296.4
XS Rating Curve= 0 ,0
Exp/Cntr(USF)=0,0
Exp/Cntr=0.3,0.1

Type RM Length L Ch R = 1 ,5268    ,150.2,148.8,146.7
XS GIS Cut Line= 3
2182306.87640913487657.4280843422182481.13738358487724.369800137
2182705.33900315487761.559642245
#Sta/Elev= 30
       0 3268.23    18.5 3259.56    82.8 3238.24    95.7 3231.45   106.1 3227.61
   125.7 3217.06   138.5 3208.51   142.8 3207.26   155.7 3200.03   177.1 3197.13
   185.6 3195.06   201.9 3195.58     206 3195.01   214.1  3193.2   224.63189.046
   230.3 3188.64   247.83189.153   250.6 3189.33   254.6  3191.1   266.5 3200.55
   270.8 3202.46   287.1 3205.86   295.2 3210.49   307.3 3218.89   318.7 3224.28
   327.6 3230.14   336.1 3233.59   351.9 3242.24   374.3 3252.93   413.9 3270.14
#Mann= 3 ,-1,0
       0      .1       0   224.6    .045       0   247.8      .1       0
Bank Sta=224.6,247.8
XS Rating Curve= 0 ,0
Exp/Cntr(USF)=0,0
Exp/Cntr=0.3,0.1

Type RM Length L Ch R = 1 ,5120    ,97.2,112,124
XS GIS Cut Line= 3
2182288.97126755487798.6113706772182418.87701812487874.137144647
2182709.56589522487891.200918617
#Sta/Elev= 30
       0 3246.44    40.7 3234.99    71.5 3221.87      87 3216.63   100.6 3210.14
   119.4 3203.52   135.9 3199.08   165.4 3192.51   195.6 3191.51   199.6 3190.75
   207.7    3187   231.7 3185.22   243.7 3182.87   259.8 3182.13   267.9 3182.85
   271.9 3184.35   283.8 3194.01   299.8 3205.68   328.5 3224.57   343.9 3233.81
   347.9 3235.78   355.9 3237.08   363.9 3241.73     376 3247.49     384 3250.33
     392 3254.94     400 3257.68     416 3266.05     424 3269.13   441.5 3278.47
#Mann= 3 ,-1,0
       0      .1       0   243.7    .045       0   267.9      .1       0
Bank Sta=243.7,267.9
XS Rating Curve= 0 ,0
Exp/Cntr=0.3,0.1

Type RM Length L Ch R = 1 ,5008    ,146.8,130.7,120
XS GIS Cut Line= 4
 2182267.6541806487822.4639051152182434.92165677487901.915956293
2182532.14587729488039.9116241272182632.50636298488042.002467579
#Sta/Elev= 30
       0 3244.99    13.9 3241.08    27.1 3239.68    49.3 3234.63    65.5 3228.48
    84.7 3219.19   106.9 3211.03   120.1 3204.42   124.6 3203.04   146.7 3197.68
   164.6 3195.42   203.8  3188.7   225.7 3183.72   237.2 3182.16   254.4 3181.26
   262.6 3179.61   271.7  3178.8   280.3  3179.6   316.4 3179.04   331.1 3177.77
   347.1 3184.53     358 3193.52     370 3208.85     374 3212.93     386 3217.82
     398  3227.2     406    3230     426 3240.76     442 3245.56   454.4 3251.07
#Mann= 3 ,-1,0
       0      .1       0   262.6    .045       0   280.3      .1       0
#XS Ineff= 2 , 0
                          320.56         3184.05
Permanent Ineff=
       F       F
Bank Sta=262.6,280.3
XS Rating Curve= 0 ,0
Exp/Cntr(USF)=0,0
Exp/Cntr=0.3,0.1

Type RM Length L Ch R = 1 ,4877    ,125.3,124,127.4
XS GIS Cut Line= 3
2182238.87212642487988.948962565 2182390.8191956488080.329717459
2182626.70905126488085.642552046
#Sta/Elev= 30
       0 3228.93    23.7 3222.72    57.5 3210.75    68.2  3208.2    82.7 3202.79
    94.9  3199.7   143.9 3189.25   164.9 3186.21   183.4  3180.1     199 3171.56
   208.73169.111   222.7 3167.86   226.7  3168.1   230.3 3169.15   242.7 3172.23
   254.7 3172.39   258.7 3171.36   270.7  3171.9   306.7 3182.86   310.7 3185.41
   314.7 3189.58   326.7 3204.03   334.7 3210.09   338.7 3212.01   346.7 3214.49
   366.7 3228.94   378.7 3234.66   390.8 3238.62   406.7 3246.74   413.3 3248.69
#Mann= 3 ,-1,0
       0      .1       0   208.7    .045       0   230.3      .1       0
Bank Sta=208.7,230.3
XS Rating Curve= 0 ,0
Exp/Cntr(USF)=0,0
Exp/Cntr=0.3,0.1

Type RM Length L Ch R = 1 ,4753    ,106.6,100.5,106.2
XS GIS Cut Line= 4
2182190.58569096488195.3553805682182314.00858607488203.312113136
2182512.15782002 488183.835906382182628.20967969488147.579607689
#Sta/Elev= 30
       0 3268.21    17.6 3259.66    33.7 3253.29    45.7 3247.04    73.7 3230.46
    89.8 3223.37    97.8 3217.79   125.9 3201.78   137.9 3197.79   150.5 3191.96
   174.1 3174.44   178.1 3168.69   182.1 3166.15   194.2 3165.37   206.2 3165.36
   242.4 3167.76   250.5 3167.05   262.5 3163.59   282.6 3162.13   286.6 3162.96
   302.7 3173.22   322.8 3176.53   335.4  3180.5   363.2 3193.16   368.9  3196.2
   398.2 3216.27   410.8 3223.79   427.6 3235.87   436.7 3240.27   444.4 3245.62
#Mann= 3 ,0,0
       0      .1       0   194.2    .045       0   206.2      .1       0
#XS Ineff= 2 , 0
                          281.52         3176.71
Permanent Ineff=
       F       F
Bank Sta=194.2,206.2
XS Rating Curve= 0 ,0
Exp/Cntr(USF)=0,0
Exp/Cntr=0.3,0.1

Type RM Length L Ch R = 1 ,4652    ,101.5,101,101.4
XS GIS Cut Line= 3
2182203.96050808488299.3908015122182369.53270636488299.029260561
2182652.32697298 488213.87299855
#Sta/Elev= 30
       0 3266.71    20.2  3255.8    60.2 3237.87    88.2 3220.75    96.2 3217.39
   108.2 3209.93   148.2 3192.17   160.2 3185.58   185.2 3177.82   197.6 3177.18
   205.9 3175.49   222.6 3169.37   235.2 3162.76  253.47 3156.08   260.2 3155.27
   271.9 3156.13     288 3160.43     302 3160.91   306.2  3162.2   318.7 3172.56
   338.5 3183.01   352.1 3191.36   360.5 3198.43     373 3204.49   385.6 3213.13
   398.1 3218.66   410.6 3226.39   423.2 3231.42   435.7  3238.5   460.9 3249.17
#Mann= 3 ,0,0
       0      .1       0  253.47    .045       0   271.9      .1       0
Bank Sta=253.47,271.9
XS Rating Curve= 0 ,0
Exp/Cntr=0.3,0.1

Type RM Length L Ch R = 1 ,4551    ,163.6,173,182.6
XS GIS Cut Line= 2
2182294.12560612488425.6639656082182662.83632645488316.219573118
#Sta/Elev= 30
       0 3212.35    18.8 3199.86    31.3 3196.91    43.9    3190    60.6 3184.73
    81.4  3176.6    93.9 3173.26   111.4 3170.38   127.3 3169.04     144 3169.54
   160.7 3167.98   180.3 3152.24   185.4 3149.28   189.9 3148.69   204.7 3149.21
   219.1 3151.99   227.5 3155.37   235.8 3155.28   244.1 3152.88   248.3 3153.65
   252.5 3155.81   259.4 3161.91   288.4 3184.45   302.6 3197.19   319.2 3210.15
   339.1 3224.17   356.8 3235.77   362.4 3238.02     372 3240.19   384.6 3247.04
#Mann= 3 ,-1,0
       0      .1       0   185.4    .045       0   204.7      .1       0
Bank Sta=185.4,204.7
XS Rating Curve= 0 ,0
Exp/Cntr(USF)=0,0
Exp/Cntr=0.3,0.1

Type RM Length L Ch R = 1 ,4378    ,108.4,105.9,101.7
XS GIS Cut Line= 2
2182301.56357454488491.5431144862182695.77590089488549.984294942
#Sta/Elev= 30
       0 3201.34     6.7 3195.99    14.8 3194.09      35 3182.76    43.1 3180.95
    75.4 3168.49    95.6 3164.65   107.8 3160.04   119.8 3156.74   140.1 3156.06
   156.3 3157.93   160.3 3157.39   168.4 3155.05   184.6 3145.75   196.7 3145.46
     208 3140.71     221 3139.59   241.2 3140.66   245.3 3141.63   250.3 3145.85
   262.3 3156.81   273.6 3168.48   281.9 3175.99   289.7 3181.54   306.6 3191.26
     318 3196.85   338.3 3203.97   350.4 3209.31   390.5 3223.07   398.5 3226.37
#Mann= 3 ,0,0
       0      .1       0     208    .045       0   241.2      .1       0
Bank Sta=208,241.2
XS Rating Curve= 0 ,0
Exp/Cntr(USF)=0,0
Exp/Cntr=0.3,0.1

Type RM Length L Ch R = 1 ,4272    ,97.4,102.2,106.1
XS GIS Cut Line= 2
2182302.17647721488631.4525756922182707.64217145488623.916038624
#Sta/Elev= 30
       0 3194.35      22  3182.7      38 3177.33      50 3172.15      70  3166.5
      94 3163.56   101.6 3161.78     138 3149.66     150 3149.31     154 3147.92
     166 3139.36     182  3138.5     190 3134.81     202 3133.15     210 3132.61
     238 3133.09     242  3133.6     254 3137.74     258 3140.07     266 3147.01
     274 3151.68     281 3156.98     294 3171.09     298 3173.74   318.1 3181.34
     334 3188.69   346.1 3191.41   378.1 3203.22   398.1 3212.08   405.5 3213.81
#Mann= 3 ,-1,0
       0      .1       0     202    .045       0     238      .1       0
Bank Sta=202,238
XS Rating Curve= 0 ,0
Exp/Cntr(USF)=0,0
Exp/Cntr=0.3,0.1

Type RM Length L Ch R = 1 ,4170    ,109.5,97.2,85.9
XS GIS Cut Line= 3
2182306.87640913 488696.618529542182548.07909937488731.683237814
2182676.64969638488678.554891945
#Sta/Elev= 30
       0 3192.68    21.5  3185.3    41.7 3180.45    53.9 3176.78      70 3169.88
    94.3 3165.22   106.4 3160.82   122.6 3156.25   130.7 3151.59   146.8 3138.51
   154.9 3135.52     167 3133.13   181.6 3125.41   187.2 3124.15   191.3 3123.95
   199.4 3123.98   206.3 3125.24   227.7 3131.01   239.8 3137.11   248.2 3139.44
   271.2 3138.66   291.5 3138.75   308.8 3140.45   313.1 3142.09   316.2 3144.12
   326.1 3152.02   339.1 3157.61     352 3165.87   368.2 3174.46   382.9 3180.23
#Mann= 3 ,-1,0
       0      .1       0   181.6    .045       0   206.3      .1       0
Bank Sta=181.6,206.3
XS Rating Curve= 0 ,0
Exp/Cntr(USF)=0,0
Exp/Cntr=0.3,0.1

Type RM Length L Ch R = 1 ,4073    ,147.8,145.5,146.4
XS GIS Cut Line= 3
2182372.75555801488848.5655987262182493.88818659488835.814795717
2182703.21386931488697.681096458
#Sta/Elev= 30
       0 3180.15    15.5 3173.58    23.5 3171.48    35.6  3165.3    51.7  3160.2
    64.4 3153.76    83.9  3146.9    97.2 3139.09     112 3127.62   116.1 3126.14
   133.8 3124.07   139.8 3121.09   143.7 3119.82   148.5 3120.05   153.23119.468
   162.8 3118.47   172.5 3119.33   182.1 3121.77   194.6 3127.35   201.2 3129.55
   214.9 3131.01     230 3135.29   273.1 3134.95   286.4 3136.75   301.9 3142.73
     313 3152.07   329.9 3162.49   335.4  3164.1   344.8 3169.62   372.6 3182.77
#Mann= 3 ,-1,0
       0      .1       0   153.2    .045       0   172.5      .1       0
Bank Sta=153.2,172.5
XS Rating Curve= 0 ,0
Exp/Cntr(USF)=0,0
Exp/Cntr=0.3,0.1

Type RM Length L Ch R = 1 ,3928    ,126,130.8,139.1
XS GIS Cut Line= 3
2182397.13684426488978.1332808052182540.33104855 488984.16251046
2182807.12446074488774.646779978
#Sta/Elev= 30
       0 3191.88     9.7 3185.55    19.1 3177.87    43.1 3164.94    63.1 3158.17
    75.1 3151.91    95.1  3143.5   111.1 3137.95   131.2 3133.19   143.3 3128.06
   163.5 3122.32   168.6 3121.72   188.9 3124.08   199.1 3123.99   204.2 3122.01
   212.9 3116.81   229.6 3116.15   251.8 3112.65     265 3109.58   270.3  3109.4
   287.8 3109.53   295.7 3110.06   305.9 3114.26   347.6 3144.46   366.9 3155.09
   374.8 3160.52   427.4 3180.93   453.4 3191.57   464.4  3196.9   482.5 3203.86
#Mann= 3 ,-1,0
       0      .1       0     265    .045       0   287.8      .1       0
Bank Sta=265,287.8
XS Rating Curve= 0 ,0
Exp/Cntr(USF)=0,0
Exp/Cntr=0.3,0.1

Type RM Length L Ch R = 1 ,3797    ,174,174.7,175.3
XS GIS Cut Line= 3
2182406.66945728489026.1831307552182574.15634294489021.575531296
 2182866.6162974488975.047811268
#Sta/Elev= 30
       0 3197.52    13.5 3188.96    25.5 3175.69    41.5 3166.51    53.5 3156.96
    57.5 3154.98    77.5 3145.47   101.5 3138.18   113.5 3135.92   125.6 3130.75
   145.6 3124.75   161.6 3117.78   193.9 3118.28   214.1 3116.16   222.2 3110.97
   226.3 3109.82   253.5 3110.76   270.9 3107.91   287.1 3110.12   305.9 3106.69
   323.6 3105.22   335.7 3104.66   341.33105.166   355.9 3114.45   388.3 3143.05
   400.7 3153.09     420 3165.44   432.9 3177.55   449.2 3187.46   463.7 3194.47
#Mann= 3 ,-1,0
       0      .1       0   323.6    .045       0   341.3      .1       0
#XS Ineff= 2 , 0
          287.96 3125.47
Permanent Ineff=
       F       F
Bank Sta=323.6,341.3
XS Rating Curve= 0 ,0
Exp/Cntr(USF)=0,0
Exp/Cntr=0.3,0.1

Type RM Length L Ch R = 1 ,3622    ,177.1,176.3,175.7
XS GIS Cut Line= 3
2182491.76305275489175.8362092792182741.46627834489162.022839354
 2182885.9753791489115.269894989
#Sta/Elev= 30
       0  3161.3    12.4  3154.5    60.5 3134.85    78.8 3131.24    84.5 3129.28
    96.6  3123.2   108.6 3114.27   116.8 3110.25   132.6 3105.51     151    3103
   164.7  3099.3   172.7 3099.21   184.7 3100.73   188.5 3100.09   196.7 3095.43
   204.7 3093.63   216.7  3092.9   226.9 3093.65   257.1 3107.22     274 3112.04
   286.6 3116.48   313.3 3128.12   322.8  3132.7   329.1 3136.77   345.4 3143.65
   353.8 3150.89   362.2 3156.65   374.9 3162.21   395.8 3172.96     402 3175.38
#Mann= 3 ,-1,0
       0      .1       0   204.7    .045       0   226.9      .1       0
Bank Sta=204.7,226.9
XS Rating Curve= 0 ,0
Exp/Cntr(USF)=0,0
Exp/Cntr=0.3,0.1

Type RM Length L Ch R = 1 ,3446    ,165,158.9,148.5
XS GIS Cut Line= 2
2182492.09721131489351.9455193622182912.63597969489327.828600746
#Sta/Elev= 30
       0 3165.64    12.1 3157.04    32.1 3147.24    44.4 3142.06    56.2  3138.3
    76.2 3133.32    96.2 3125.93   104.2 3123.91   120.4 3116.91   132.3 3114.61
   140.3 3112.07   152.3 3106.97   180.4  3090.2   196.4 3085.46   200.4 3084.89
   228.5 3084.69   241.4 3085.41   252.5 3086.55   256.6 3089.03   268.5 3098.48
   280.5 3106.43   284.5 3108.84   288.6 3110.28   316.6 3115.86   336.6 3118.75
   349.9 3122.25   364.7 3124.07   388.7 3128.71   404.7 3133.06   421.2 3136.29
#Mann= 3 ,-1,0
       0      .1       0   196.4    .045       0   241.4      .1       0
Bank Sta=196.4,241.4
XS Rating Curve= 0 ,0
Exp/Cntr(USF)=0,0
Exp/Cntr=0.3,0.1

Type RM Length L Ch R = 1 ,3287    ,126.9,136.9,147.6
XS GIS Cut Line= 3
2182545.95396554 489463.791843892182703.21386931489505.231953668
2182917.85238662489434.039970203
#Sta/Elev= 30
       0  3136.9    18.8 3133.25      23 3131.85    80.9 3105.12    97.4  3100.1
   109.8 3097.97   138.8 3096.84   155.3 3097.47   159.5 3097.02   164.1 3094.95
   172.1 3089.84   180.5 3086.76   188.9 3082.19   191.9 3081.14   201.4 3081.39
   205.8 3080.85   226.3 3075.39   235.3 3074.33   256.4 3075.45   274.2 3086.92
   277.4 3089.84   281.6 3095.03   286.9 3100.23   296.3 3106.45   306.9 3112.39
   323.8 3117.18   353.3 3121.65   361.7  3123.5   365.9 3125.54   388.8 3131.95
#Mann= 3 ,-1,0
       0      .1       0   226.3    .045       0   256.4      .1       0
Bank Sta=226.3,256.4
XS Rating Curve= 0 ,0
Exp/Cntr(USF)=0,0
Exp/Cntr=0.3,0.1

Type RM Length L Ch R = 1 ,3150    ,157.5,159.2,161
XS GIS Cut Line= 3
2182548.07909937489534.9838273542182847.72297008489628.489716084
2182939.10372497489619.989180745
#Sta/Elev= 30
       0 3131.99    16.9 3126.02    33.8 3118.62      42 3116.07    54.6 3109.72
    88.1 3096.49     109  3092.1     130 3091.91   150.9 3089.06   155.2 3087.73
   167.7 3079.54   171.9  3078.1   176.1  3077.3   192.9 3078.77   201.2 3076.19
   205.4 3075.64     218 3075.58   251.5 3067.49   255.7 3066.99   272.5 3067.47
   280.8 3068.52   301.8 3074.87   310.2 3080.07   338.5  3100.4   350.4  3110.9
   358.5 3117.14   366.6 3121.91   378.6 3124.85   398.7 3135.38   405.7 3136.95
#Mann= 3 ,-1,0
       0      .1       0   251.5    .045       0   272.5      .1       0
Bank Sta=251.5,272.5
XS Rating Curve= 0 ,0
Exp/Cntr(USF)=0,0
Exp/Cntr=0.3,0.1

Type RM Length L Ch R = 1 ,2991    ,221.9,211.9,207
XS GIS Cut Line= 3
2182492.70013428489648.8850798292182827.77457231489800.821667113
2182937.65728276 489804.89139713
#Sta/Elev= 30
       0 3137.11    12.6 3133.78    75.4 3112.59   100.4  3101.9   113.6 3094.47
   132.8 3085.18     140 3082.09   153.9 3078.09     163 3073.99   170.7 3069.07
   175.1 3067.58   201.5 3063.79     219 3066.17   232.2 3065.35   236.6  3064.7
   244.6 3058.24   262.7 3057.16  272.63  3058.2   284.9 3063.49     308 3080.42
   329.2 3081.95   346.4 3086.54   359.6 3088.74   376.3 3093.43   420.3 3108.16
   432.4 3111.36   448.4 3119.14   460.4 3122.29   468.4  3126.7   477.9 3130.27
#Mann= 3 ,-1,0
       0      .1       0   244.6    .045       0  272.63      .1       0
Bank Sta=244.6,272.63
XS Rating Curve= 0 ,0
Exp/Cntr(USF)=0,0
Exp/Cntr=0.3,0.1

Type RM Length L Ch R = 1 ,2779    ,135,139.4,141.8
XS GIS Cut Line= 3
2182411.57850476489905.5178460552182668.69804015489945.881413176
2182880.03039181489943.829224596
#Sta/Elev= 30
       0 3149.48    16.8 3138.31    28.9  3131.3    42.2 3125.42    65.4 3116.38
    77.5  3110.8    93.7  3105.4   105.9 3102.49     118 3097.88   129.7 3094.79
   146.4 3088.06   174.7 3072.09   178.8 3068.53   186.9 3059.76   196.2 3051.88
     199 3050.47   207.7 3050.15   223.3  3048.9   239.5 3050.12   247.6 3053.34
   263.1  3054.1   267.7 3055.27   280.3 3055.53   303.7 3059.15   319.7 3067.94
   335.8 3070.13   391.2 3088.49   431.8 3100.54   451.8 3105.24   471.6 3112.38
#Mann= 3 ,0,0
       0      .1       0   207.7    .045       0   239.5      .1       0
Bank Sta=207.7,239.5
XS Rating Curve= 0 ,0
Exp/Cntr(USF)=0,0
Exp/Cntr=0.3,0.1

Type RM Length L Ch R = 1 ,2640    ,126.3,121.3,115.4
XS GIS Cut Line= 3
2182448.19780914490022.702042433 2182666.0240272490094.956592815
2182859.41120617 490072.64268755
#Sta/Elev= 30
       0 3121.65    21.3  3111.9    33.6 3105.33    49.4 3100.62    71.6 3091.94
      80 3086.62    96.9 3077.54   113.8 3064.33   128.5 3054.92     139 3044.67
   143.3 3041.27   147.5 3039.56   155.9 3038.56     173 3039.45   185.4 3040.34
   201.3 3044.93   210.7 3044.36   219.1 3046.55   229.4  3046.7   243.7 3050.19
   267.9 3053.28   292.1 3053.41   311.9 3061.55   324.3 3069.28   332.3 3073.39
   340.4 3075.43   348.4 3078.67   372.6 3083.97   388.3  3089.7   424.2 3097.11
#Mann= 3 ,-1,0
       0      .1       0   147.5    .045       0     173      .1       0
Bank Sta=147.5,173
XS Rating Curve= 0 ,0
Exp/Cntr(USF)=0,0
Exp/Cntr=0.3,0.1

Type RM Length L Ch R = 1 ,2518    ,143.9,131,115.2
XS GIS Cut Line= 2
2182452.00283411490192.8723253742182894.24682925490175.236828636
#Sta/Elev= 30
       0 3113.71    16.2 3106.49    44.2 3096.72    60.2 3090.29    76.9 3082.14
    84.2 3076.38    92.2 3064.34   108.3 3036.83   110.7 3035.16   112.3 3034.12
   116.3 3033.91   124.3 3034.02   130.8 3034.93   144.3 3036.33   165.4 3036.25
   204.3 3038.52   208.3 3038.22   216.3 3040.57   232.4 3041.04   244.4 3043.48
   284.4 3046.65   296.3 3051.81   308.4 3059.34   316.4 3062.33   376.5 3075.92
   396.5 3083.61   404.5 3085.83   415.6  3091.1   424.5 3094.47   442.6 3100.18
#Mann= 3 ,-1,0
       0      .1       0   110.7    .045       0   130.8      .1       0
Bank Sta=110.7,130.8
XS Rating Curve= 0 ,0
Exp/Cntr(USF)=0,0
Exp/Cntr=0.3,0.1

Type RM Length L Ch R = 1 ,2387    ,130.1,155.8,183.2
XS GIS Cut Line= 4
2182502.38872193490290.4689056132182654.33579111490298.969440952
2182701.08873548490216.0892213962182880.66254452490201.213284553
#Sta/Elev= 30
       0 3090.22    25.8 3082.27    29.8 3080.19    41.9 3075.76    49.9 3072.07
    57.9 3069.58    69.9 3063.61    93.9 3053.98   117.8 3041.27     130 3035.74
     142  3033.4   166.6 3030.34   176.33028.195   181.8 3027.77   188.5 3028.21
   198.9  3029.7   209.4 3033.06   219.4    3034   227.7 3033.75   237.3 3038.62
   254.5 3040.52   274.5  3047.6   282.5 3051.31   298.6 3056.83   322.7 3060.57
   330.7 3063.15   342.8 3065.27   358.8 3070.28   370.9 3072.26   427.5 3093.22
#Mann= 3 ,-1,0
       0      .1       0   176.3    .045       0   188.5      .1       0
Bank Sta=176.3,188.5
XS Rating Curve= 0 ,0
Exp/Cntr(USF)=0,0
Exp/Cntr=0.3,0.1

Type RM Length L Ch R = 1 ,2231    ,109.5,106.6,107.6
XS GIS Cut Line= 3
2182467.02427783490320.4525128362182650.58255071490343.397296946
2182895.80493089  490438.0445314
#Sta/Elev= 30
       0  3103.2     9.2 3098.27    25.3 3092.93    37.4 3086.44    53.6 3083.07
    65.7 3077.38    89.8 3068.81     102 3065.69   146.3 3051.45   162.4 3049.21
   187.6 3039.69   208.1 3035.55   212.4 3033.76     221 3028.15   233.5 3023.88
   246.7 3021.82   263.9 3023.63   271.1 3022.37   276.7 3021.72  304.13 3022.43
   314.4 3025.49   319.6 3026.33   328.2 3029.88   342.3 3037.45   359.2 3047.94
     367 3052.01   385.6 3055.28   413.4  3062.9   431.1 3068.38   447.8 3076.12
#Mann= 3 ,-1,0
       0      .1       0   271.1    .045       0  304.13      .1       0
Bank Sta=271.1,304.13
XS Rating Curve= 0 ,0
Exp/Cntr(USF)=0,0
Exp/Cntr=0.3,0.1

Type RM Length L Ch R = 1 ,2125    ,92,89.8,88.9
XS GIS Cut Line= 3
2182508.76412343490442.4159747982182785.03152195490492.356619915
2182894.47591444490487.043785328
#Sta/Elev= 30
       0 3081.54    15.7 3076.34    32.9 3069.84      40 3066.74    48.2 3063.97
    56.3 3060.35    77.6 3052.47     101 3046.06   109.2 3043.41   137.6 3037.42
   170.1 3023.89   174.5 3021.69  186.09 3014.83   190.4 3014.05   198.6 3014.79
   202.6 3015.04   206.7  3016.3   215.3  3016.9   231.1 3019.04   239.2 3018.19
   243.3 3020.06   251.4 3025.54   263.5 3031.89   280.7 3039.46   283.9 3040.56
   299.9  3044.2   328.8 3049.84     336 3051.73   360.7 3059.97   390.3 3072.08
#Mann= 3 ,-1,0
       0      .1       0  186.09    .045       0   198.6      .1       0
#XS Ineff= 2 , 0
                          231.67         3027.62
Permanent Ineff=
       F       F
Bank Sta=186.09,198.6
XS Rating Curve= 0 ,0
Exp/Cntr(USF)=0,0
Exp/Cntr=0.3,0.1

Type RM Length L Ch R = 1 ,2035    ,134.3,132.6,130.5
XS GIS Cut Line= 3
2182489.98698094490557.791450191 2182808.7824989490571.357216913
2182914.59547933490544.225683469
#Sta/Elev= 30
       0 3082.95    14.2 3077.95    26.2 3074.98    50.2 3066.52      74 3059.27
    78.3 3058.57   101.4 3050.55   124.4 3040.55   150.3 3028.01   174.4 3019.83
   182.4 3014.22   191.1 3009.93   198.4 3009.41   214.4 3009.97   222.4 3012.04
   230.4 3012.14   234.4 3013.21   258.4 3025.67   278.4  3034.6   286.4 3036.78
   310.5 3040.32   322.6 3045.07   333.5 3050.84   351.5 3057.45     368 3060.49
   379.5 3064.38   396.9 3068.48     401 3069.78   409.3 3075.21   428.3 3078.88
#Mann= 3 ,-1,0
       0      .1       0   191.1    .045       0   214.4      .1       0
Bank Sta=191.1,214.4
XS Rating Curve= 0 ,0
Exp/Cntr(USF)=0,0
Exp/Cntr=0.3,0.1

Type RM Length L Ch R = 1 ,1902    ,133.4,129.3,126.8
XS GIS Cut Line= 3
 2182482.1999505490659.1796259442182647.96038961490702.744869557
2182853.03580466490681.493531209
#Sta/Elev= 30
       0  3084.1    23.6 3074.82    35.1 3068.09    47.5 3058.76    59.9 3052.37
    68.2 3046.75    84.1 3039.56      93 3037.77    97.2 3036.17   109.6 3029.67
   117.8 3026.53   126.1 3021.95   138.5 3016.97   163.3 3009.41   167.5 3008.46
   179.6 3007.58   203.8 3001.61   209.4 3001.24   219.2 3001.62   231.9 3002.67
   235.9 3005.77     244 3014.53     248 3016.73     252 3017.75   260.1 3018.39
   272.1 3021.34   288.2 3022.11   308.3 3028.11   340.5 3033.78   377.6 3037.54
#Mann= 3 ,-1,0
       0      .1       0   203.8    .045       0   219.2      .1       0
Bank Sta=203.8,219.2
XS Rating Curve= 0 ,0
Exp/Cntr(USF)=0,0
Exp/Cntr=0.3,0.1

Type RM Length L Ch R = 1 ,1773    ,114.2,112.9,112.9
XS GIS Cut Line= 3
2182510.88925727 490827.06519889 2182666.0240272490839.816001899
2182871.09944226490767.561451517
#Sta/Elev= 30
       0 3071.27    13.3 3065.94    21.4 3062.17    33.4 3059.14    45.4 3054.01
    53.5 3049.78    61.5 3046.49    69.5 3042.36    77.8 3039.45    81.6  3037.3
    93.6  3029.1   101.6 3025.76   113.7 3018.15   121.7 3014.47   129.7 3010.21
   143.4 3003.99   159.4 2999.04   162.2 2998.54   170.7 2998.26   188.1 2994.84
   200.2 2994.32   207.2 2994.96   215.9 2996.33     230 3001.55   238.5 3004.24
   271.9 3021.95   285.2 3027.63   289.4 3028.98   316.2 3033.43   373.1  3041.3
#Mann= 3 ,-1,0
       0      .1       0   188.1    .045       0   207.2      .1       0
Bank Sta=188.1,207.2
XS Rating Curve= 0 ,0
Exp/Cntr(USF)=0,0
Exp/Cntr=0.3,0.1

Type RM Length L Ch R = 1 ,1660    ,195.4,205.6,215
XS GIS Cut Line= 3
2182540.92821597490952.2199340412182630.46227634490973.925160795
2182950.61437097490854.546413643
#Sta/Elev= 30
       0 3052.67    15.7 3045.63    32.2 3040.08    44.5 3034.72    98.2 3016.06
   106.8 3011.41   117.2 3007.95   123.8 3004.78   128.1 3003.71     158 3003.15
   162.3 3000.99   170.8 2993.74   175.1 2991.31   208.8 2989.57   219.72987.934
   226.3 2987.47   231.6 2987.97   247.6 2989.29   256.2 2990.62   264.7 2993.38
   273.3 2997.58   277.6 3000.29   298.9 3016.18   303.1 3019.87   311.6 3025.53
   315.9 3027.84   320.2 3029.32   330.4 3030.48   401.3 3042.06   433.8 3049.44
#Mann= 3 ,-1,0
       0      .1       0   219.7    .045       0   231.6      .1       0
#XS Ineff= 2 , 0
          182.55 3001.67
Permanent Ineff=
       F       F
Bank Sta=219.7,231.6
XS Rating Curve= 0 ,0
Exp/Cntr(USF)=0,0
Exp/Cntr=0.3,0.1

Type RM Length L Ch R = 1 ,1455    ,116.5,112.4,102.7
XS GIS Cut Line= 4
2182502.18698244491043.5965105872182628.79916926491067.989684194
2182798.38980481491149.3002628842182918.03251345491142.330784711
#Sta/Elev= 30
       0 3053.82     6.1 3050.64    18.3 3046.44    34.6 3038.59    50.9 3032.83
    83.5 3017.43    87.6 3014.94    99.8 3004.72   116.1 2994.12   128.3 2988.62
   132.7 2987.28   159.3 2985.66   168.3 2986.94   171.3 2986.65   189.3 2981.39
   207.3 2980.49   218.8 2978.84   230.3 2977.46   239.1  2978.6     248 2979.08
   264.3 2984.15   270.5 2985.45   314.6  2983.2   334.8 2986.94   338.8 2987.89
   346.9 2991.39     368 3001.78   386.9 3009.99     419 3019.03   436.9 3022.76
#Mann= 3 ,-1,0
       0      .1       0   218.8    .045       0   239.1      .1       0
Bank Sta=218.8,239.1
XS Rating Curve= 0 ,0
Exp/Cntr(USF)=0,0
Exp/Cntr=0.3,0.1

Type RM Length L Ch R = 1 ,1342    ,91.6,90.5,88.1
XS GIS Cut Line= 3
2182482.44012761491167.8855380132182645.83525577491207.464155313
2182904.09355711491205.056088271
#Sta/Elev= 30
       0 3041.42    22.4 3030.32    30.6 3028.08    47.1 3021.25    75.9 3012.39
    88.2 3007.67   108.8 3003.08   129.4 2987.32   149.9 2973.17   154.9 2970.38
   161.5 2969.31   174.5 2971.91 186.5052971.679   194.5 2970.49206.50492971.651
   230.5  2974.8   242.5 2979.09   262.5 2977.48   274.5 2979.58   293.3 2976.41
   302.5 2975.82   325.7 2978.42   338.5  2977.2   358.5 2982.67   370.5 2987.18
   382.5 2993.91   394.5 2999.46   406.5 3007.02   418.5 3011.41   426.4 3013.26
#Mann= 3 ,-1,0
       0      .1       0 186.505    .045       0206.5049      .1       0
Bank Sta=186.505,206.5049
XS Rating Curve= 0 ,0
Exp/Cntr(USF)=0,0
Exp/Cntr=0.3,0.1

Type RM Length L Ch R = 1 ,1252    ,90.4,89.2,86.5
XS GIS Cut Line= 4
2182486.45021817491280.7812726122182606.52027983491306.282878629
2182712.77697157491290.3443748692182867.91174151491244.653997421
#Sta/Elev= 30
       0  3024.1     9.9 3020.82    30.4 3012.68    38.6 3011.31    71.3  2999.2
    79.5 2993.47    99.9  2982.2   116.3 2968.94   124.4  2965.2   136.6 2961.81
   148.7 2961.21   160.8 2959.04   168.9 2959.64   178.52958.368   185.1 2957.59
   194.8 2958.85   209.4 2961.58   227.2 2968.56   233.5 2968.52   246.2 2967.02
   269.3 2968.56   283.8 2970.86   300.5 2970.75   304.6 2970.18   329.6  2974.4
   346.3 2976.52     363 2981.55   375.6  2987.7   383.9 2993.32   391.9 2997.54
#Mann= 3 ,-1,0
       0      .1       0   178.5    .045       0   194.8      .1       0
Bank Sta=178.5,194.8
XS Rating Curve= 0 ,0
Exp/Cntr(USF)=0,0
Exp/Cntr=0.3,0.1

Type RM Length L Ch R = 1 ,1163    ,141.4,142.7,144.1
XS GIS Cut Line= 3
2182500.74599052491393.3952000722182566.01632053 491420.09669871
2182845.88758404491330.102758855
#Sta/Elev= 30
       0 3010.89    16.7 3004.56    38.3 2993.28    46.9 2989.47    70.5  2985.3
    89.6 2982.97      98 2980.44   102.2 2978.65   110.6 2973.08   125.4 2960.81
   135.8 2956.67   144.2 2956.09   152.6 2957.05   173.6 2955.62   177.8 2954.84
   186.2 2951.33   194.6 2949.23   198.8 2948.16   207.2    2949   215.6 2949.56
   236.7 2948.71   245.1 2952.52   249.3 2953.18   257.7 2953.21   261.9 2954.78
   273.7 2962.22   303.9 2979.09   309.8 2981.73   341.6 2993.23   364.5 2997.86
#Mann= 3 ,-1,0
       0      .1       0   194.6    .045       0   207.2      .1       0
Bank Sta=194.6,207.2
XS Rating Curve= 0 ,0
Exp/Cntr(USF)=0,0
Exp/Cntr=0.3,0.1

Type RM Length L Ch R = 1 ,1020    ,95.8,100.9,104.9
XS GIS Cut Line= 4
2182501.32615501 491476.293585412182691.52563322491521.983962858
2182798.84489188491501.7951914282182866.84917459491458.229947815
#Sta/Elev= 30
       0 2991.63    27.6  2985.6    56.4  2981.8    81.1  2976.4   101.7 2968.43
     114  2962.3   122.5 2959.13   138.7 2951.08   142.8 2950.42   155.1 2951.23
   167.5 2946.75   175.7 2944.83   216.6 2944.74   220.7 2943.43   228.8  2939.1
   234.5 2938.14   245.5 2939.01   251.7 2940.37   264.9 2939.75   269.5 2940.53
   273.6 2942.74   281.7 2952.01   285.8 2954.97     294 2959.87   314.9 2974.22
   338.1 2987.03   344.4 2989.15   353.9 2990.46   372.8 2995.01   385.6 2997.22
#Mann= 3 ,-1,0
       0      .1       0   228.8    .045       0   245.5      .1       0
Bank Sta=228.8,245.5
XS Rating Curve= 0 ,0
Exp/Cntr(USF)=0,0
Exp/Cntr=0.3,0.1

Type RM Length L Ch R = 1 ,919     ,135.7,137.8,135.9
XS GIS Cut Line= 4
2182510.88925727491567.6743403052182686.21279863491605.926749331
2182778.65612045491619.7401192572182854.09837158491608.051883166
#Sta/Elev= 30
       0 2978.27    13.6 2976.15    29.2  2975.4    38.2 2973.99    49.4 2973.24
    54.5 2972.07    62.7 2968.79      75 2966.31    83.2 2963.48    91.4 2959.11
    99.6 2955.64   107.8 2950.53     116 2947.54   128.2 2946.32   136.4 2944.37
   148.7  2943.7     161 2940.24   169.2 2939.35   197.6 2938.71   205.7 2935.77
   215.7  2934.1   225.9 2933.36     234  2934.1   250.2 2937.73   254.4 2940.37
     286 2964.28   298.7 2972.37   310.9  2977.9   331.1 2983.37   349.3 2991.49
#Mann= 3 ,-1,0
       0      .1       0   215.7    .045       0     234      .1       0
Bank Sta=215.7,234
XS Rating Curve= 0 ,0
Exp/Cntr(USF)=0,0
Exp/Cntr=0.3,0.1

Type RM Length L Ch R = 1 ,781     ,134.9,143.1,150
XS GIS Cut Line= 3
2182468.11082552491684.1448519142182548.21532144491719.746850099
 2182868.6333051491759.304625859
#Sta/Elev= 30
       0  2971.7    30.7 2967.42      57 2960.32    61.4 2958.36    87.7 2940.77
   103.7 2933.73   111.8 2932.46     132 2931.44     136 2931.66     144 2934.57
   152.1 2935.17   168.2 2930.63   184.3 2933.56   200.1 2932.04   212.6 2932.64
   220.6 2931.08   228.7 2926.89   242.3 2926.17   248.8 2925.76   253.9 2926.18
     269 2929.19   281.1 2933.89   285.1 2936.02   297.2 2945.44   318.5 2960.41
   349.6 2972.73   361.6 2974.26   375.9 2977.35   393.9 2979.56   410.5 2983.16
#Mann= 3 ,-1,0
       0      .1       0   242.3    .045       0   253.9      .1       0
Bank Sta=242.3,253.9
XS Rating Curve= 0 ,0
Exp/Cntr(USF)=0,0
Exp/Cntr=0.3,0.1

Type RM Length L Ch R = 1 ,638     ,164.6,163.1,160.7
XS GIS Cut Line= 4
2182462.01117907491761.0615192692182618.20851592491840.754038072
2182698.96360164491917.2588561242182761.65504977491917.258856124
#Sta/Elev= 30
       0 2963.81    11.4 2962.54    38.4 2956.52    49.3  2952.3    65.3 2944.58
    74.3 2938.84    90.9 2930.83    96.8 2928.46   105.7 2926.16   114.7 2928.18
   119.2  2928.5   123.7 2928.33   137.1 2925.15   146.1 2925.63   156.3 2927.19
   173.1 2924.93   181.8 2925.14   188.4 2923.34  198.28 2916.78   200.1 2916.09
   215.7 2916.79   233.2 2917.96   238.7 2919.65   263.2 2942.79   276.1 2952.32
   281.7  2954.6   303.8 2956.53   319.9 2956.28   331.8 2957.04   349.3 2960.17
#Mann= 3 ,-1,0
       0      .1       0  198.28    .045       0   215.7      .1       0
Bank Sta=198.28,215.7
XS Rating Curve= 0 ,0
Exp/Cntr(USF)=0,0
Exp/Cntr=0.3,0.1

Type RM Length L Ch R = 1 ,475     ,88.7,81.9,78.9
XS GIS Cut Line= 3
2182349.43749824491856.2211764742182588.76204159492019.397001487
 2182703.4795913492049.065333308
#Sta/Elev= 30
       0 2976.02    17.8 2969.36    48.7 2960.95    58.5 2957.15    68.9 2954.74
    80.4  2950.8    90.5 2945.86   100.1 2939.34   114.9 2930.41     138  2921.9
   148.6 2919.14   157.9 2920.42   163.1 2919.88   172.8 2915.69   193.4 2908.42
     197 2907.89     207 2908.23   215.7 2907.62  222.75 2908.36     226 2909.75
   232.9 2914.57   235.7 2915.82   244.5 2917.27   257.3  2922.4   284.1 2941.07
   288.9 2943.98   293.2 2945.42   310.3 2946.67   388.2 2947.25   408.2 2948.45
#Mann= 3 ,-1,0
       0      .1       0     207    .045       0  222.75      .1       0
Bank Sta=207,222.75
XS Rating Curve= 0 ,0
Exp/Cntr(USF)=0,0
Exp/Cntr=0.3,0.1

Type RM Length L Ch R = 1 ,393     ,82.4,82.9,82.9
XS GIS Cut Line= 4
2182316.65625482 491963.870373162182394.01746254492028.686520173
2182607.28349465492072.5942326652182706.59855862492070.503389213
#Sta/Elev= 30
       0 2958.65    77.3 2944.41    98.5 2939.08   107.2 2936.08   119.5 2934.98
   123.5 2933.71     144 2918.91   148.1 2917.23   160.3  2916.2   164.4  2915.1
   172.6 2908.35   177.7 2906.71   188.9  2905.2   201.1  2904.7   204.8  2905.2
   225.6 2908.42     242 2909.76   246.1 2911.36   258.3 2920.87   266.5 2925.64
   270.6 2927.41   278.7 2928.64   282.7 2930.03   293.3 2936.16   303.2 2940.64
   315.5 2943.54   330.7 2945.02   351.6 2945.62   383.6 2944.92     418 2947.67
#Mann= 3 ,-1,0
       0      .1       0   188.9    .045       0   204.8      .1       0
Bank Sta=188.9,204.8
XS Rating Curve= 0 ,0
Exp/Cntr(USF)=0,0
Exp/Cntr=0.3,0.1

Type RM Length L Ch R = 1 ,310     ,103.5,102,102.8
XS GIS Cut Line= 4
 2182317.5020783492046.8920200442182431.19673846492119.146570426
2182521.51492644492140.3979087742182698.96360164492124.459405013
#Sta/Elev= 30
       0 2950.29    11.7 2948.07    22.1 2944.66    35.5 2943.49      50 2938.55
    83.7  2931.7      98 2927.36   116.9 2914.39   121.7 2913.44   135.7 2912.66
   156.3 2899.93   160.2 2899.07   172.7 2898.58   181.7 2899.03   189.1 2900.13
   197.4 2899.29   217.9 2909.99     222 2911.71   226.1 2912.32   230.2 2912.56
   242.2 2910.34   270.3 2910.51   282.4 2912.07   291.9 2915.39   297.5 2918.26
   321.4 2933.99   330.6  2940.8   334.6 2942.17   358.7 2941.58   405.7 2944.93
#Mann= 3 ,-1,0
       0      .1       0   160.2    .045       0   181.7      .1       0
Bank Sta=160.2,181.7
XS Rating Curve= 0 ,0
Exp/Cntr(USF)=0,0
Exp/Cntr=0.3,0.1
